--- FshCrk.prj (project) ---

Proj Title=FshCrk
Current Plan=p01
Default Exp/Contr=0,0
English Units
Geom File=g01
Flow File=f01
Plan File=p01
BEGIN DESCRIPTION:
---------- MODELED AS PART OF WVEM CTP PROGRAM, 2025----------
Stream Name: Fish Creek
Flood Zone: AFH
Marshall County, WV
HEC-RAS Version: RAS 6.6
Vertical Datum: NAVD88
Projection: NAD 1983 StatePlane West Virginia N FIPS 4701 (US Feet)
Terrain: 1-meter West Virginia FEMA R3 South Central (collected 2018-2019)
Land Use: 2024 NLCD
Hydrologic Method:
Duda et al., "Estimation of magnitude and frequency of floods for rural, unregulated streams in and near Virginia and West Virginia." September 8, 2025.
Additional Model Notes:
KWSE to Zone AE
END DESCRIPTION:
DSS Export Rating Curves= 0
DSS Export Rating Curve Sorted= 0
DSS Export Volume Flow Curves= 0
DXF OffsetX= 0
DXF OffsetY= 0
DXF ScaleX= 0
DXF ScaleY= 0

--- FshCrk.p01 (plan) ---

Plan Title=Floodplain
Program Version=6.60
Short Identifier=Floodplain
Geom File=g01
Flow File=f01
Subcritical Flow
K Sum by GR= 0
Std Step Tol= 0.01
Critical Tol= 0.01
Num of Std Step Trials= 20
Max Error Tol= 0.3
Flow Tol Ratio= 0.001
Split Flow NTrial= 30
Split Flow Tol= 0.02
Split Flow Ratio= 0.02
Log Output Level= 0
Friction Slope Method= 1
Unsteady Friction Slope Method= 2
Unsteady Bridges Friction Slope Method= 1
Parabolic Critical Depth
Global Vel Dist= 0 , 0 , 0
Global Log Level= 0
CheckData=False
Encroach Param=-1 ,0,0, 0
Flow Ratio Tolerance=0.1
Flow Ratio Min Ratio=0.5
Flow Ratio Max Ratio=4
Flow Ratio Max Iterations= 10
Mapping Interval=1HOUR
Computation Time Step Use Courant=        0
Computation Time Step Use Time Series=    0
Computation Time Step Count To Double=0
Computation Time Step Max Doubling=0
Computation Time Step Max Halving=0
Computation Time Step Residence Courant=0
Run HTab= 0
Run UNet= 0
Run Sediment= 0
Run PostProcess= 0
Run WQNet= 0
Run RASMapper=-1
UNET Theta= 0
UNET Theta Warmup= 0
UNET ZTol= 0
UNET ZSATol= 0
UNET MxIter= 0
UNET Max Iter WO Improvement= 0
UNET MaxInSteps= 0
UNET DtIC= 0
UNET DtMin= 0
UNET MaxCRTS= 0
UNET WFStab= 0
UNET SFStab= 0
UNET WFX= 1
UNET SFX= 1
UNET Gravity=32.17405
UNET 1D Methodology=Finite Difference
UNET DSS MLevel= 1
UNET Pardiso=0
UNET DZMax Abort= 0
UNET Use Existing IB Tables= 0
UNET Froude Reduction=False
UNET Froude Limit= 0
UNET Froude Power= 0
UNET D1 Cores= 0
UNET WindReference=Eulerian
UNET WindDragFormulation=Hsu (1988)
UNET D2 Coriolis=0
UNET D2 Cores= 0
UNET D2 Theta= 1
UNET D2 Theta Warmup= 1
UNET D2 Z Tol= 0.01
UNET D2 Volume Tol= 0.01
UNET D2 Max Iterations= 20
UNET D2 Advanced Convergence=0
UNET D2 WS Max Tol=0.15
UNET D2 WS RMS Tol=0.002
UNET D2 WS Stall Tol=1
UNET D2 Equation= 0
UNET D2 RampUpFraction=0.1
UNET D2 TimeSlices= 1
UNET D2 Turbulence Formulation=Non-Conservative (original)
UNET D2 Eddy Viscosity=0.3
UNET D2 Transverse Eddy Viscosity=0.1
UNET D2 Smagorinsky Mixing=0
UNET D2 BCVolumeCheck=0
UNET D2 Cores=0
UNET D2 SolverType=PARDISO (Direct)
UNET D2 Minimum Iterations= 3
UNET D2 Maximum Iterations= 30
UNET D2 Restart Number= 10
UNET D2 Relaxation Coeff=1.3
UNET D2 SOR Precondition Iterations= 10
UNET D2 ILUT Maximum Fill= 8
UNET D2 ILUT Tolerance=1E-08
UNET D2 Convergence Tolerance=0.00001
PS Theta= 1
PS WS Tol= 0.01
PS Volume Tol= 0.01
PS Max Iterations= 20
PS Equation= 0
PS Advance Time Step=-1
PS Target Courant=0.9
PS Time Slices= 1
PS Iterate With 2D=0
PS Project Initial WSE from DS=-1
PS Ramp Up Initial WSE from US=-1
PS Cores=0
UNET D1D2 MaxIter= 0
UNET D1D2 ZTol=0.01
UNET D1D2 QTol=0.1
UNET D1D2 MinQTol=1
Write IC File= 0
Write IC File at Fixed DateTime=0
Write IC File at Sim End=0
Echo Input=False
Echo Parameters=False
Echo Output=False
Write Detailed= 0
HDF Write Warmup=0
HDF Write Time Slices=0
HDF Flush=0
HDF Compression= 1
HDF Chunk Size= 1
HDF Spatial Parts= 1
HDF Use Max Rows=0
HDF Fixed Rows= 1
Calibration Method= 0
Calibration Iterations= 20
Calibration Max Change=0.05
Calibration Tolerance=0.2
Calibration Maximum=1.5
Calibration Minimum=0.5
Calibration Optimization Method= 1
WQ AD Non Conservative
WQ ULTIMATE=-1
WQ Max Comp Step=1HOUR
WQ Output Interval=15MIN
WQ Output Selected Increments= 0
WQ Create Restart=0
WQ Fixed Restart=0
WQ System Summary=0
WQ Write To DSS=0
Sorting and Armoring Iterations= 10
XS Update Threshold= 0.02
Bed Roughness Predictor= 0
Processes Affected by Predictor=Sediment Only
Hydraulics Update Threshold= 0.02
Energy Slope Method= 1
Volume Change Method= 1
Sediment Retention Method= 0
Sediment TS Multiplier= 1
Warm Up Method= 0
XS Weighting Method= 0
Number of US Weighted Cross Sections= 1
Number of DS Weighted Cross Sections= 1
Upstream XS Weight=0
Main XS Weight=1
Downstream XS Weight=0
Number of DS XS's Weighted with US Boundary= 1
Upstream Boundary Weight= 1
Weight of XSs Associated with US Boundary= 0
Number of US XS's Weighted with DS Boundary= 1
Downstream Boundary Weight= 0.5
Weight of XSs Associated with DS Boundary= 0.5
Percentile Method= 0
Sediment Output Level= 3
Mass or Volume Output= 0
Output Increment Type= 1
Profile and TS Output Increment= 1
Transport Output Increment 1
XS Output Flag= 0
XS Output Increment= 10
Read HDF5 Sediment Hotstart= 0
Sediment Hotstart Type= 0
Write Gradation File= 0
Read Gradation Hotstart= 0
Write HDF5 File= 1
Write Binary Output= 1
Write DSS Sediment File= 0
DSS Sediment Output Type= 1
SV Curve= 0
Specific Gage Flag= 0
Subcell Erosion Methods= 0
Subcell Deposition Methods= 0
Advection Scheme= 1
Matrix Solver= 0
Implicit Weighting Factor= 1
Maximum Outer Loop Convergence Iterations= 5
Convergence Maximum Absolute= 0.001
Convergence RMSE= 0.0001
Grain Fractions Max Abs Error= 0.001
Max Subgrid Regions= 1
Max Subgrid Length Scale= 3.402823E+38
Initial Layer Thickness= 3
Min Layer Thickness= 0.1
Max Layer Thickness= 6
Number of Layers= 5

--- FshCrk.f01 (steady flow) ---

Flow Title=Flow
Program Version=6.60
Number of Profiles= 1
Profile Names=P100yr
River Rch & RM=FshCrk,Main,137849
    9920
River Rch & RM=FshCrk,Main,105902
   13600
River Rch & RM=FshCrk,Main,90818
   15200
River Rch & RM=FshCrk,Main,52152
   17400
Boundary for River Rch & Prof#=FshCrk,Main            , 1
Up Type= 0
Dn Type= 1
Dn Known WS=644
DSS Import GetInterval= 0
DSS Import GetPeak= 0
DSS Import FillOption= 0

--- FshCrk.g01 (geometry) ---

Geom Title=Geometry
Program Version=6.60

River Reach=FshCrk          ,Main
Reach XY= 30
     1666630.542      446628.978     1665595.164      448172.373
     1663389.371      445250.597     1662145.833      447909.722
     1664806.945        453387.5     1662690.278        454912.5
     1659819.444      452109.722     1661049.098      458549.058
     1658078.889      457941.111       1656838.4        460147.2
     1654994.792      458190.972     1651899.306       463227.43
     1646705.247       462538.58     1646527.778      465410.397
     1641411.111      465828.889     1642140.445      468630.044
     1640689.236       462741.32     1636223.958      462800.347
     1635827.778      465306.667      1632946.18      465359.375
        1632140.      469945.555     1627552.626      462497.287
      1628834.93      467768.661      1624906.25      465972.222
        1625250.      470725.694     1621020.833      468571.181
     1621865.167      475273.132     1619749.599      475088.755
     1618677.775      471687.3171615975.85636511473390.112471268

Type RM Length L Ch R = 1 ,137849  ,380.1,395.4,403.4
XS GIS Cut Line= 6
1665929.46459681446649.4938098941666226.86459255446647.392764226
1666580.24905638446640.7008484751666680.22064123  446643.0804369
1667032.88594639446666.5846549721667329.84893514446682.837903306
#Sta/Elev= 30
       0  1024.5    34.1 1008.92     126  977.46     313  934.54   470.5  885.72
   559.1  874.48   647.7  871.24   654.3  868.26   669.8849.1772   677.2  847.44
   734.5849.1591   785.6  872.45     904  892.43   936.9  905.83   950.1  912.78
   979.7  937.44  1021.9  976.81    1068  991.43  1084.9 1005.72  1094.7 1023.19
  1117.7 1022.03  1137.4 1029.45  1147.3 1036.46  1173.6 1065.45    1190 1090.04
  1222.9 1120.77  1245.9 1147.94    1259 1172.66    1328 1227.42  1401.7  1268.2
#Mann= 3 ,-1,0
       0      .1       0   669.8    .045       0   734.5      .1       0
Bank Sta=669.8,734.5
XS Rating Curve= 0 ,0
Exp/Cntr(USF)=0,0
Exp/Cntr=0.3,0.1

Type RM Length L Ch R = 1 ,137454  ,490.6,491.4,491.1
XS GIS Cut Line= 6
1665892.96824914446741.8810478431666652.24100882447065.575938506
1666730.09649615 447106.072576671666899.20672223447196.373577176
1666987.52773981447241.3104951811667167.09529406447329.438927842
#Sta/Elev= 30
       0 1027.26    48.3 1006.12    80.4   998.1   112.4  982.55   205.2  954.25
   312.2  935.07   490.5  882.37   554.9  872.89   647.4  867.19     669849.0118
   675.9  847.58   725.7848.9935     740  850.49   769.9  863.68   833.2  871.53
   884.9   893.5   936.4  942.11   948.8  960.84     963  974.29    1004  983.77
  1018.9  992.66  1037.4 1011.08  1070.1 1016.93  1085.7 1024.17  1107.9 1047.78
  1133.7 1083.36  1183.3 1120.07  1210.9 1146.21  1258.5 1172.78    1404  1219.6
#Mann= 3 ,-1,0
       0      .1       0     669    .045       0   725.7      .1       0
Bank Sta=669,725.7
XS Rating Curve= 0 ,0
Exp/Cntr(USF)=0,0
Exp/Cntr=0.3,0.1

Type RM Length L Ch R = 1 ,136962  ,597.5,611.9,624.6
XS GIS Cut Line= 6
1665758.96057655447085.6148491491665805.97459014447225.849148734
1665985.15959922447309.6337580671666073.39826788 447349.70749682
1666159.22552406447387.4561089861667000.57751589447741.709993644
#Sta/Elev= 30
       0 1073.98    38.8 1073.58   147.9 1063.28   195.3 1052.34   217.1 1042.63
   264.2 1013.98   293.1 1006.37   318.4  988.61   361.7  974.79   409.5  938.05
   430.1   930.6   455.3  911.41   501.9  888.01   586.4  860.04   656.6  853.87
   681.4847.6542   736.7  847.12   772.8  847.66   896.5  912.56   964.9  957.39
  1012.3  964.19  1096.6  984.14  1142.5 1011.14    1184 1024.01  1235.2 1062.22
  1287.8 1090.26    1353 1106.58  1406.3 1130.66  1428.1 1146.21  1449.3 1154.66
#Mann= 3 ,-1,0
       0      .1       0   681.4    .045       0   772.8      .1       0
Bank Sta=681.4,772.8
XS Rating Curve= 0 ,0
Exp/Cntr(USF)=0,0
Exp/Cntr=0.3,0.1

Type RM Length L Ch R = 1 ,136351  ,388.8,429.9,435.2
XS GIS Cut Line= 6
1665677.12028523447231.199011311 1665692.4493228447416.707170472
 1665718.8193488447549.8033609841665766.82220556447642.893397897
1665878.63070898 447797.352734641666431.49443264448523.789601982
#Sta/Elev= 30
       0  1056.3   102.8 1030.91   148.9 1010.07   181.8 1003.48   208.5  988.47
   228.6  982.34   288.8  972.64   333.3  956.37   445.5  940.29   515.4  922.96
   550.7  908.46   611.3   868.8     649  851.44   693.5  853.04   742.7  845.15
  816.72845.0816     828  844.56   850.4  845.09   904.2  872.15  1017.6  896.97
  1071.8     918  1120.5  941.28  1151.8  964.57  1221.9  989.38  1254.9 1008.59
  1308.5 1025.09  1320.9 1040.87  1380.6 1077.25  1501.2 1130.77  1530.2 1149.72
#Mann= 5 ,-1,0
       0      .1       0  754.78     .06       0  764.78      .1       0
  816.72    .045       0   850.4      .1       0
Bank Sta=816.72,850.4
XS Rating Curve= 0 ,0
Exp/Cntr(USF)=0,0
Exp/Cntr=0.3,0.1

Type RM Length L Ch R = 1 ,135921  ,520.5,569,582.7
XS GIS Cut Line= 3
1665663.07306921 447236.265930311665652.53814048447501.952141958
1665712.56635299448694.755001843
#Sta/Elev= 30
       0 1052.89   110.6 1010.13   146.7 1003.56   199.2  980.24   248.5  970.92
   289.4  952.18   317.5  943.96   466.1  924.12   540.8  905.75   636.1  904.67
     721  867.44   744.5  863.25   866.1  861.44  892.44 843.166   938.3   842.2
   971.2  843.16   971.2  843.17  1018.1  867.18  1090.1  882.56    1137  898.88
    1188  940.65  1217.5     976    1257  982.84  1302.7 1011.57  1332.5 1020.26
  1339.1 1026.09  1348.9 1043.86  1381.8 1081.67  1424.5 1101.59  1460.2 1109.21
#Mann= 5 ,-1,0
       0      .1       0  795.89     .06       0  855.89      .1       0
  892.44    .045       0   971.2      .1       0
Bank Sta=892.44,971.2
XS Rating Curve= 0 ,0
Exp/Cntr(USF)=0,0
Exp/Cntr=0.3,0.1

Type RM Length L Ch R = 1 ,135352  ,339.3,354.2,371.2
XS GIS Cut Line= 6
1665644.56129523447222.670156971 1665627.3313428  447399.6497899
1665588.58306073 447515.688599811665448.93701455447653.678481311
 1665270.4363873447839.154160231 1664804.0396823448427.002065897
#Sta/Elev= 30
       0 1050.86    25.8 1043.13    98.3 1009.47   144.5  999.95   181.4  982.93
   233.3  969.45   277.3  948.43   558.1  880.46   729.9  861.92     764 843.157
   845.2   841.9   850.9  843.17   895.3  864.72   965.4  872.48  1018.6  897.89
  1063.5  934.72  1085.4  962.49  1131.3  975.16  1152.4  996.77    1200 1020.18
  1227.5 1050.67    1237  1069.4  1244.2  1078.3  1306.9 1123.56  1336.1 1141.96
  1365.4 1153.66  1381.2 1167.17  1457.3  1216.8  1475.5 1222.19  1504.3 1217.39
#Mann= 3 ,-1,0
       0      .1       0     764    .045       0   850.9      .1       0
Bank Sta=764,850.9
XS Rating Curve= 0 ,0
Exp/Cntr(USF)=0,0
Exp/Cntr=0.3,0.1

Type RM Length L Ch R = 1 ,134997  ,641.4,646.9,651.2
XS GIS Cut Line= 6
1665618.65227567447235.4622989021665564.11444296447302.126377793
1664766.80501395447734.5658016221664595.11867754447827.682741377
1664506.51452404447872.4274025431664416.18104328447914.941097039
#Sta/Elev= 30
       0 1037.94    56.2 1001.69    81.1  995.44   101.9  978.88   180.1  957.98
   214.2  937.37     243  927.13     400  900.95     439  886.73   507.2  871.59
   527.4  857.25   545.5  851.29   654.6842.9758   723.4  842.17   731.1842.9857
   747.6  856.94     773  859.33   803.6  873.74   840.9  912.04     867  930.77
   896.4  959.59   932.7  973.42   949.2  993.56   985.9 1012.18  1049.9 1075.37
  1120.8 1109.83  1145.6 1137.66  1184.3 1167.67  1242.4 1189.59  1387.6 1227.53
#Mann= 3 ,-1,0
       0      .1       0   654.6    .045       0   731.1      .1       0
Bank Sta=654.6,731.1
XS Rating Curve= 0 ,0
Exp/Cntr(USF)=0,0
Exp/Cntr=0.3,0.1

Type RM Length L Ch R = 1 ,134351  ,486.1,478.8,459
XS GIS Cut Line= 6
 1665440.0521898446842.7473603931665336.68133356446851.566568479
1665234.54767956446861.0324288161665135.18567355446875.832924142
1665042.38041297446904.0927101371664096.35441789447248.127127066
#Sta/Elev= 30
       0 1050.91    60.8 1039.03   123.2 1023.16   172.6    1006   238.8  990.52
   280.9  971.64   325.6  958.86     415  899.46   428.9  887.42   512.7  842.81
     586  840.73     600  845.82   639.7  845.87   676.8840.4014   701.2  839.94
   740.5840.4078     813  866.59   865.3  895.29   893.1   916.1   914.2  925.88
   959.4  959.02   994.5  968.36  1010.9  976.61  1036.2   995.3  1056.9 1001.21
  1130.6 1056.53  1148.1 1072.76  1207.4 1103.31  1256.3 1114.16  1410.4 1121.48
#Mann= 3 ,-1,0
       0      .1       0   676.8    .045       0   740.5      .1       0
Bank Sta=676.8,740.5
XS Rating Curve= 0 ,0
Exp/Cntr(USF)=0,0
Exp/Cntr=0.3,0.1

Type RM Length L Ch R = 1 ,133872  ,507.8,500,488.3
XS GIS Cut Line= 6
1665241.83900355446116.953536391 1665084.4131373446238.401784316
1665006.47333255446298.5292887241664929.77073005446357.702726811
1664647.70272464446575.3072784841664059.82506197446990.961984842
#Sta/Elev= 30
       0 1006.46    11.4 1017.12    25.4 1041.13    49.7 1069.96   101.3 1103.83
   128.3 1133.59     145 1140.79   176.5 1134.67   231.2 1099.46   334.2 1060.69
     423 1008.21   472.4  988.54   495.5  969.09   530.4  957.66   588.4  910.59
   654.6  847.06   669.5838.9003   696.7  837.82   745.7838.8906   814.3  848.41
   939.2   850.3  1023.6  886.12  1127.7  953.45  1169.5  967.31    1196  988.93
    1226 1000.28  1264.3 1029.58  1301.3 1050.25  1352.7  1060.5  1470.4  1067.7
#Mann= 3 ,-1,0
       0      .1       0   669.5    .045       0   745.7      .1       0
Bank Sta=669.5,745.7
XS Rating Curve= 0 ,0
Exp/Cntr(USF)=0,0
Exp/Cntr=0.3,0.1

Type RM Length L Ch R = 1 ,133372  ,507.2,500,498.1
XS GIS Cut Line= 6
1664782.01183923445650.1280264711664715.27608031445724.423153475
1664649.44812797445798.9285818931664585.43677305 445873.85461314
1664525.05828489445949.6225062311663907.87185521446744.862057477
#Sta/Elev= 30
       0 1195.12   141.7 1127.72   176.7  1098.9   201.5 1090.66   215.6  1078.8
   239.4 1068.14   346.6  995.95   372.3  988.85   397.5  972.55   468.9  949.38
   510.4  921.98   564.4   903.3   594.4  883.14   626.7  854.55   669.4838.6245
   693.1  837.48   745.8838.6082   783.8   846.3   855.1  846.17     889  857.47
   959.4  894.57    1045  952.18    1076  965.36  1087.8  966.97  1116.7  988.16
  1158.3 1007.95  1209.3 1037.38  1245.5 1039.76  1291.2 1035.34  1401.4 1044.61
#Mann= 3 ,-1,0
       0      .1       0   669.4    .045       0   745.8      .1       0
Bank Sta=669.4,745.8
XS Rating Curve= 0 ,0
Exp/Cntr(USF)=0,0
Exp/Cntr=0.3,0.1

Type RM Length L Ch R = 1 ,132872  ,478.9,500,512.2
XS GIS Cut Line= 6
1664390.65140148445276.938812226 1664322.2178113445350.977049977
1664259.33604731445428.2692182211663755.30884014 446179.54527472
1663645.18766931446343.6837259831663589.50569406446427.790841222
#Sta/Elev= 30
       0 1158.43    33.5 1134.52    75.2 1114.04    93.3 1097.24   112.5 1093.15
     146 1073.98   182.4 1063.08   231.1 1027.06   266.7 1005.47   307.6  986.59
   327.3  970.32   392.7  947.99   428.7  923.65     518  883.01   543.3  881.91
   560.6  874.29   574.7  860.86   594.6  849.57   626.2  839.35   646.2837.7502
   681.5  837.41   738.8837.7482   833.7  855.76   879.1  879.51   941.2  923.13
   993.6  943.91  1098.7  965.06  1228.2 1000.32  1298.3 1015.07  1403.7 1048.06
#Mann= 3 ,-1,0
       0      .1       0   646.2    .045       0   738.8      .1       0
Bank Sta=646.2,738.8
XS Rating Curve= 0 ,0
Exp/Cntr(USF)=0,0
Exp/Cntr=0.3,0.1

Type RM Length L Ch R = 1 ,132372  ,567,500,428
XS GIS Cut Line= 6
1664235.59232838445053.0960840581663586.82569564445523.813570341
1663456.92123457445730.7486465081663437.28093289446013.528874472
1663459.47216147446184.0925097321663496.64794014446347.995397151
#Sta/Elev= 30
       0  1172.4    80.9 1172.24   112.6 1165.54   140.6 1153.08   187.5 1125.26
   215.8 1100.51     243 1089.33   258.1 1077.08     313 1048.21   386.8  997.35
   409.8  988.09   430.9  970.98   475.6  955.31     552  912.09   593.8  879.77
   609.5  863.56   646.6  836.84   684.7  835.84     746  836.84   755.1  842.12
   787.4  848.88   899.6  845.44   913.9  852.78   944.8  877.03   966.7  885.09
  1004.3   890.6  1103.7  893.24  1248.4  917.24  1479.9  968.75  1669.4 1023.32
#Mann= 3 ,-1,0
       0      .1       0   646.6    .045       0     746      .1       0
Bank Sta=646.6,746
XS Rating Curve= 0 ,0
Exp/Cntr(USF)=0,0
Exp/Cntr=0.3,0.1

Type RM Length L Ch R = 1 ,131872  ,524.2,500,473.2
XS GIS Cut Line= 6
1662866.14034289444739.4067508131663341.39464173445414.242671475
1663368.61210696445508.5466167331663421.34625347446003.552844554
1663451.50498581446179.104658812 1663492.6643523446345.501307637
#Sta/Elev= 30
       0  977.36    25.6  974.38    40.6  967.33   103.2  972.02   145.6  962.28
   171.5  961.86   200.1  980.01   243.7  972.75   279.8  983.15   338.7  991.78
   392.9  990.15   433.7  970.63   512.6  949.63   520.6  942.06   532.6  918.99
   584.8   856.6   616.5  838.09   659.2836.1287   685.1  835.57   742.4 836.123
   805.5  848.78   931.1     845   944.3  847.36   967.4  861.68   990.4  869.41
  1254.4   893.6  1366.6  917.05  1462.7   943.8  1550.1  959.59  1770.9 1022.33
#Mann= 5 ,-1,0
       0      .1       0  645.39     .08       0   659.2    .045       0
   742.4     .08       0  750.39      .1       0
Bank Sta=659.2,742.4
XS Rating Curve= 0 ,0
Exp/Cntr(USF)=0,0
Exp/Cntr=0.3,0.1

Type RM Length L Ch R = 1 ,131372  ,500.3,500,499.3
XS GIS Cut Line= 6
1662324.06006221445492.4062290641663279.08374272445810.611629397
1663349.72303714 445903.15475139 1663395.8161208446046.781760722
1663438.73991947446200.7191168961663486.28181913446356.308372647
#Sta/Elev= 30
       0 1159.88   178.7 1171.65   219.1 1166.64   230.6 1156.57   250.2 1126.86
     279 1101.54   299.8 1091.35   315.3 1075.13   336.1 1067.19   353.9 1051.49
   364.6 1036.58   395.4 1018.75   440.4   986.2     458  965.81   485.3  951.45
   509.5  919.61     558  868.97   589.1  858.46   630.6  851.51   663.1  834.11
   713.6  833.37   739.8834.1106   758.9  840.26   796.6  836.86   848.4  838.45
     883  858.82  1082.7  885.94  1264.4  938.29  1373.5  960.11  1596.4 1026.41
#Mann= 4 ,-1,0
       0      .1       0   663.1    .045       0   739.8     .08       0
  740.39      .1       0
Bank Sta=663.1,739.8
XS Rating Curve= 0 ,0
Exp/Cntr(USF)=0,0
Exp/Cntr=0.3,0.1

Type RM Length L Ch R = 1 ,130872  ,481.7,482.2,482.2
XS GIS Cut Line= 6
 1662139.4524918445952.0398242321662684.28440739446137.060451567
1662921.00703105446217.4497264771663092.63070355 446275.73209022
1663371.51958147446370.4405622331663452.67165014446441.169423386
#Sta/Elev= 30
       0 1165.27    36.8 1145.47   102.6 1095.26   151.1 1074.22   185.8 1062.08
   283.8 1001.96   348.5  975.69   386.7  957.82   428.7  945.27     456  930.91
   487.2  917.94   525.3  905.15   577.3  893.27   608.5  872.44   636.2  843.53
   646.6  835.88   654.8833.2123   674.3  832.59   753.7  833.22   785.2  839.16
   795.9  843.57   878.8  843.88   923.8  857.56   961.9  874.07  1086.6  958.42
  1103.7  963.07  1168.4  992.91  1239.1 1012.08  1301.2 1023.89  1408.8 1057.42
#Mann= 3 ,-1,0
       0      .1       0   654.8    .045       0   753.7      .1       0
Bank Sta=654.8,753.7
XS Rating Curve= 0 ,0
Exp/Cntr(USF)=0,0
Exp/Cntr=0.3,0.1

Type RM Length L Ch R = 1 ,130390  ,516.1,517.8,521.7
XS GIS Cut Line= 2
1662029.70685679 446422.266259871663318.48996927446852.721752807
#Sta/Elev= 30
       0 1053.49    33.3 1032.08    55.6 1021.53      80 1003.01   121.5  985.38
   147.4  968.54   200.9  950.95     246  930.74   321.9  913.68     398  908.62
   436.1   901.2   584.8  852.51   619.3  832.05   686.8   831.3695.5208832.0846
   754.2  833.37   792.3  851.04   826.3  861.31   844.2  862.99     865  871.28
   899.6  892.77   961.8  949.05  1005.7  964.63    1055  998.89  1079.4 1024.22
  1092.1 1033.77  1120.9 1046.51  1148.3 1051.88  1239.1 1048.59  1358.8 1055.37
#Mann= 3 ,-1,0
       0      .1       0   619.3    .045       0695.5208      .1       0
Bank Sta=619.3,695.5208
XS Rating Curve= 0 ,0
Exp/Cntr(USF)=0,0
Exp/Cntr=0.3,0.1

Type RM Length L Ch R = 1 ,129872  ,495.9,500,503.2
XS GIS Cut Line= 6
1661893.95856021446862.8381994811661987.66998698446897.403419063
1662080.67931539446932.5677188041662172.28444713446968.930178896
1662261.08085747447007.6896158161663177.18105939447424.925001815
#Sta/Elev= 30
       0  878.37    22.5   882.2      75  880.71     138  871.54   208.3  869.23
   246.8   863.8   401.9  849.93   525.8  846.84   580.6  837.64   620.2  836.11
   634.7  832.24   671.2829.5168   698.3  828.86   736.9829.5086     750  834.55
   760.8  841.07   778.9  846.47   793.3  856.75   818.5  883.39   854.6  916.82
   865.4  934.47   877.5  949.16   896.2  959.05   939.4  969.99   995.2  980.08
  1081.7 1001.23    1179 1033.05  1229.5 1043.95  1305.2 1050.33  1401.4 1050.32
#Mann= 5 ,-1,0
       0      .1       0  646.01     .08       0   671.2    .045       0
   736.9     .08       0  741.01      .1       0
Bank Sta=671.2,736.9
XS Rating Curve= 0 ,0
Exp/Cntr(USF)=0,0
Exp/Cntr=0.3,0.1

Type RM Length L Ch R = 1 ,129372  ,550.3,500,450.5
XS GIS Cut Line= 6
1661712.04324163447231.6586560611662583.07069905447736.278053641
1662678.03277947447764.7839021381662805.67983389 447736.61958839
1662949.42396897447675.9517307281663091.72552164447608.193007976
#Sta/Elev= 30
       0 1009.47    18.4   997.7    44.8  987.55    71.1   970.8    97.5  964.13
   156.4  931.84   199.6  916.41   291.1  897.38   336.3  882.92   461.5  852.54
   529.9  843.42   591.1  841.74   610.6  833.54   643.9829.0684   651.3  827.88
     732829.0715   750.4  836.87   761.4  849.68   784.2  884.67   803.2  904.55
   811.5  908.62   848.7  910.93   931.5  908.16   975.8  916.21  1021.9  920.44
  1130.8  920.05  1274.1  948.35    1388  963.25  1466.6  986.04  1550.2 1022.09
#Mann= 3 ,-1,0
       0      .1       0   643.9    .045       0     732      .1       0
Bank Sta=643.9,732
XS Rating Curve= 0 ,0
Exp/Cntr(USF)=0,0
Exp/Cntr=0.3,0.1

Type RM Length L Ch R = 1 ,128872  ,521.4,500,476.6
XS GIS Cut Line= 6
1661611.76719548448429.8130838871662290.63788497447960.317631811
1662390.04024522447920.5726325661662641.85995156447836.685989305
1662787.59325589447772.5706319811663087.20387714447617.180850893
#Sta/Elev= 30
       0 1184.65   180.4  1133.6   200.9 1123.22   218.1 1108.24   236.9  1099.2
   253.4 1085.36   279.3 1070.65   309.9 1035.59   342.9 1006.14   370.3  997.56
     390  980.07   418.3  971.04   430.1  963.51   481.2  915.84   515.6  888.75
     527  874.88     567  854.05   635.7  843.31   654.9828.7966   730.7  827.96
     743828.8046   762.7  833.52   781.5  846.94   984.8  859.96  1127.1  893.22
  1257.1  912.18  1429.9     948  1530.9  961.04    1616  984.32  1694.7 1018.08
#Mann= 3 ,-1,0
       0      .1       0   654.9    .045       0     743      .1       0
Bank Sta=654.9,743
XS Rating Curve= 0 ,0
Exp/Cntr(USF)=0,0
Exp/Cntr=0.3,0.1

Type RM Length L Ch R = 1 ,128372  ,509.7,499.9,508.5
XS GIS Cut Line= 6
1662313.36552981448903.4207324831662698.81718673448075.896796972
1662769.47944698447898.5208393931662851.40316764 447803.48789297
1662972.28579989447709.3860470651663103.15627305447624.910166144
#Sta/Elev= 30
       0   949.6    16.2  948.83    66.9  914.88   113.8  929.81   182.7  971.65
   259.5  983.32   370.9  980.34   402.7  970.01   416.5   960.6   425.2  949.64
     436  930.22   446.9  920.96   457.7  904.11   490.3  872.96     512  858.92
   559.1  847.91   585.4  834.54   637.2  828.75  720.28 828.732   750.9  831.13
   812.1  826.91   823.3  828.29   834.1  835.69   906.4  842.32   968.1  885.97
  1147.9  920.37  1217.2  937.31  1369.1  960.75  1451.9  984.78  1538.3 1022.25
#Mann= 4 ,-1,0
       0     .06       0      20      .1       0   637.2    .045       0
  720.28      .1       0
Bank Sta=637.2,720.28
XS Rating Curve= 0 ,0
Exp/Cntr(USF)=0,0
Exp/Cntr=0.3,0.1

Type RM Length L Ch R = 1 ,127872  ,490.2,500.1,514.6
XS GIS Cut Line= 6
1662831.61449331449016.2262811361662961.09487739 448625.49477914
1662992.75065397448534.7826902271663032.73745064448456.635536805
1663069.53265263448391.2567305561663421.77013713 447728.67439431
#Sta/Elev= 30
       0  907.41    37.6   909.9    86.2  920.77     197  936.44   228.1  922.94
   322.6  850.17   352.3  836.59   400.5  835.76   452.5  827.72   491.3  827.41
   515.5  832.55   656.8  826.37     679  828.48   693.2825.7789   716.5  825.03
   761.6 825.784   831.8  878.38   857.7  903.97     880  921.68     924     941
   969.2  968.92  1017.5  981.62  1047.7   996.9  1147.5 1033.55  1177.2  1038.9
  1240.4 1038.06  1281.3 1035.37  1303.5 1028.99  1329.5  1037.4  1420.9 1043.81
#Mann= 3 ,-1,0
       0      .1       0   693.2    .045       0   761.6      .1       0
Bank Sta=693.2,761.6
XS Rating Curve= 0 ,0
Exp/Cntr(USF)=0,0
Exp/Cntr=0.3,0.1

Type RM Length L Ch R = 1 ,127372  ,485.5,500,511.7
XS GIS Cut Line= 6
1662932.16678564 449103.572891221663086.84396972448978.642694891
1663379.78826572448742.0355565551663438.13362147448694.909994647
1663944.40393439448286.0010355561664021.89426497448223.412578061
#Sta/Elev= 30
       0  897.83    94.4  905.23   169.1  904.76   206.4  899.87   253.1  880.12
   303.6  840.86   324.7  833.87     519  834.57   535.1  829.58     582  825.75
   678.5824.3839   708.5  823.68   732.6824.3802     744  828.27   770.1  849.23
   792.8  877.27   806.6  903.94   826.6  927.29   852.6   950.1     883  969.71
     918  980.49   940.4  997.73   968.5 1007.75  1012.1 1038.03  1041.6 1049.61
  1104.9 1066.69  1155.5 1086.37  1230.6 1107.68  1291.2 1131.42  1400.8 1168.59
#Mann= 5 ,-1,0
       0      .1       0  585.39     .06       0  625.39      .1       0
   678.5    .045       0   732.6      .1       0
Bank Sta=678.5,732.6
XS Rating Curve= 0 ,0
Exp/Cntr(USF)=0,0
Exp/Cntr=0.3,0.1

Type RM Length L Ch R = 1 ,126872  ,194.2,181.6,168.1
XS GIS Cut Line= 6
1663010.50521164449279.8048222211663107.14051706449255.645749807
1663568.71603747449140.2522798031663641.47671872449122.062355563
1663987.09020072449035.6589850631664081.07262431449012.163625225
#Sta/Elev= 30
       0  886.33    27.4  883.82    71.4  875.24   115.4  877.61   290.3   865.2
   335.2  857.46     369  841.03   396.1   836.7   588.8  831.78   609.1  825.66
   636.2  825.41     649823.1613   690.3  822.37   721.1  823.17   768.1  836.93
   791.7  845.31   801.9   851.2   856.4  903.46   872.9  924.23   886.4  937.54
   899.9  956.42   910.1   966.6     927  978.92   947.3  982.11   961.3   988.5
   991.3 1019.19  1006.6 1039.13  1014.9 1046.46  1042.4 1056.38  1103.5 1060.01
#Mann= 3 ,-1,0
       0      .1       0     649    .045       0   721.1      .1       0
Bank Sta=649,721.1
XS Rating Curve= 0 ,0
Exp/Cntr(USF)=0,0
Exp/Cntr=0.3,0.1

Type RM Length L Ch R = 1 ,126690  ,316.3,318.4,317.8
XS GIS Cut Line= 3
1662857.30979629449504.7712761091663393.89493296449477.533451913
1664110.24970932449068.966088969
#Sta/Elev= 30
       0  881.54    33.1  879.84    68.4  870.88    97.9  866.95   166.9  861.48
   265.5  856.06     341  858.27   360.7  851.31   373.8  849.65   602.5   845.8
   670.4  839.84     814  834.93  873.01822.6167   957.4  822.28   980.1  822.69
   988.8  825.43  1002.8  835.06  1036.9   842.6  1077.8  865.79  1104.2  891.32
  1112.3  895.28  1123.7  910.98  1157.1  948.14  1183.6  972.05  1221.9  988.93
  1234.1 1002.64  1248.3 1011.97    1271 1036.45  1286.1 1040.76    1362 1044.32
#Mann= 8 ,-1,0
       0      .1       0     260     .06       0     350      .1       0
     440     .05       0  667.28      .1       0  767.28     .06       0
  873.01    .045       0   980.1      .1       0
Bank Sta=873.01,980.1
XS Rating Curve= 0 ,0
Exp/Cntr(USF)=0,0
Exp/Cntr=0.3,0.1

Type RM Length L Ch R = 1 ,126372  ,509.8,500,488.5
XS GIS Cut Line= 6
1663232.32957114449919.2133203151663736.12876038449641.254886732
1664031.63637146449478.216826975 1664113.2024813449431.986932561
1664197.08157864 449383.48079598 1664282.1174978449333.836538315
#Sta/Elev= 30
       0  860.02    80.6  856.56   181.7   847.1   272.3  843.32   406.6  842.56
   489.6  843.71   541.5  843.22   593.9  841.03   605.2  839.31   627.6  828.14
  662.82822.4432   725.1  821.19   773.8  822.43   783.8  825.11   793.5  830.86
   798.3  832.18   837.5  831.75     878   834.7   886.2  837.93   901.2  846.35
   923.8  853.44   942.6  864.73   950.6  867.41  1014.3  868.36  1030.1  872.87
  1059.7  877.12  1082.5  884.24  1099.3  885.44    1147  893.43    1202  896.71
#Mann= 9 ,-1,0
       0      .1       0      70     .06       0  179.61     .07       0
  268.83     .06       0  278.83     .05       0  575.39      .1       0
  585.39     .06       0  662.82    .045       0   773.8      .1       0
Bank Sta=662.82,773.8
XS Rating Curve= 0 ,0
Exp/Cntr(USF)=0,0
Exp/Cntr=0.3,0.1

Type RM Length L Ch R = 1 ,125872  ,521,500,485.5
XS GIS Cut Line= 6
1663623.67524514450504.0002084821664147.69158556449966.884812891
1664202.32533455449915.405257061 1664269.5761843449858.772168234
1664340.22499314449794.4681629841664628.08498172449510.091435149
#Sta/Elev= 30
       0  1038.9    43.3  1028.9    87.1 1022.16   170.7 1002.14     189 1000.97
   209.7   997.5   267.4  982.28   320.5  977.61   359.1  971.91     391  958.93
   460.7  927.21   484.9     911   536.6  882.92   592.8  843.98   615.7  834.26
   639.3  832.57   666.2  820.74   675.3  819.97  736.05820.7137   770.7  820.84
   788.7  825.84   820.3  831.88     939  828.57   957.5  829.24   987.7  833.52
  1029.5  843.72  1219.8  846.79    1301  851.09  1359.8  861.42  1413.6  881.18
#Mann= 4 ,-1,0
       0      .1       0  575.39     .06       0   666.2    .045       0
  736.05      .1       0
Bank Sta=666.2,736.05
XS Rating Curve= 0 ,0
Exp/Cntr(USF)=0,0
Exp/Cntr=0.3,0.1

Type RM Length L Ch R = 1 ,125372  ,471.3,499.9,519.9
XS GIS Cut Line= 6
1664171.06194563450854.3804132341664274.28221163450792.516035646
1664377.58876355450621.1269427241664421.51387255450534.404347137
 1664495.4576223450368.805596977 1664805.8192063449603.988228977
#Sta/Elev= 30
       0 1016.24    32.8 1004.84    51.2   990.5    82.5  983.44   120.3  967.39
   137.4  963.16   151.7  956.19   187.4  943.79   231.1  934.88   247.1  934.41
   297.9  918.28   335.3  913.37   394.2   913.2   456.1  901.75   499.5  876.67
   521.1  858.82   542.5  854.27   567.5  840.43   588.2  832.23   615.8  831.24
   644.4  820.33   737.6  819.55   761.8820.3227     787  829.21   938.2     831
   970.9  836.16  1020.9  834.57  1137.7  841.07  1345.1  862.35  1424.5  882.73
#Mann= 4 ,-1,0
       0      .1       0  541.58     .06       0   644.4    .045       0
   761.8      .1       0
Bank Sta=644.4,761.8
XS Rating Curve= 0 ,0
Exp/Cntr(USF)=0,0
Exp/Cntr=0.3,0.1

Type RM Length L Ch R = 1 ,124872  ,462.2,500.1,545.9
XS GIS Cut Line= 6
1664203.87913722 450887.82916522 1664459.3553323450841.067447722
1664565.86528988  450814.79453441664656.72271971450772.147966146
 1664866.3997938 450623.197476641665438.70704813 450137.86183314
#Sta/Elev= 30
       0 1000.97    21.4  989.34    61.6  976.95   105.1   946.3   135.8  935.15
   168.5  914.95   251.5  889.94   431.4  860.72   467.5  859.76   495.2  853.09
   535.2  850.25   551.2  841.87   574.6  840.43   595.3  827.59   607.5  824.69
     760818.5933   766.9  817.95   834.9  818.59   850.7  827.69     931  826.22
   976.4  835.08  1095.1  838.62  1197.8  856.67  1269.7  886.71  1295.3  907.04
  1344.2  937.56  1374.4  967.47  1404.3  983.86  1418.7  987.09  1477.5 1022.61
#Mann= 3 ,-1,0
       0      .1       0     760    .045       0   834.9      .1       0
Bank Sta=760,834.9
XS Rating Curve= 0 ,0
Exp/Cntr(USF)=0,0
Exp/Cntr=0.3,0.1

Type RM Length L Ch R = 1 ,124372  ,531.6,542.1,560.7
XS GIS Cut Line= 6
1664205.04448922450895.8406321411664342.24762689450875.436473474
1664464.01674031450873.1136434821664575.18876205450878.886597812
1664675.36933596450900.3320929711665538.60645464451418.164718732
#Sta/Elev= 30
       0  998.18    56.4  978.39    99.6  947.33   142.6  931.68   185.3  907.69
     310  874.32   409.4     854   659.5  834.36   678.6  824.01     738 817.332
   751.4  816.12   796.6817.3527   824.2  832.94   912.3  847.98   972.5  882.09
   985.3  885.63  1035.3  936.59  1059.2   951.7  1084.7  982.66    1123  995.57
  1138.1 1011.48  1161.3 1029.62  1180.4 1053.44  1214.1 1088.66  1264.7 1102.79
  1283.8 1113.37  1318.3 1120.24  1345.1 1140.52  1410.6  1161.1  1480.9 1202.89
#Mann= 7 ,-1,0
       0      .1       0  381.83     .05       0  578.05      .1       0
  598.05     .05       0  618.05      .1       0     738    .045       0
   796.6      .1       0
Bank Sta=738,796.6
XS Rating Curve= 0 ,0
Exp/Cntr(USF)=0,0
Exp/Cntr=0.3,0.1

Type RM Length L Ch R = 1 ,123830  ,99.9,101.1,105.5
XS GIS Cut Line= 5
1664160.83859014 450984.848224691664559.00621127 451402.48199069
1664748.10695927451664.9706591911664816.97351379451758.143056471
1665180.60796355451696.545127896
#Sta/Elev= 30
       0  977.86    36.7   978.5    64.1   974.1    82.6  968.14     145  938.16
   249.6  922.19     277  904.03   326.2  860.64   387.5  834.37   482.5  830.02
   563.4  833.01   595.7  830.81   622.6  822.71   675.7816.5117     685  815.73
   750.2816.5143   795.4  839.03   841.5  843.13   911.9  859.96  1008.1  864.02
  1024.7  868.91  1054.7  867.48  1067.5  874.51  1113.4  887.36  1197.7  907.03
  1221.6  909.38  1292.7  935.39  1314.2   947.1  1354.1  975.76  1385.2  988.64
#Mann= 5 ,-1,0
       0      .1       0     430     .05       0     550      .1       0
   675.7    .045       0   750.2      .1       0
Bank Sta=675.7,750.2
XS Rating Curve= 0 ,0
Exp/Cntr(USF)=0,0
Exp/Cntr=0.3,0.1

Type RM Length L Ch R = 1 ,123729  ,385.7,356.4,309
XS GIS Cut Line= 5
1664091.55685531451051.9098738131664489.72447644451469.543639813
1664678.82522444451732.0323083141664747.69177895451825.204705594
1665111.32622872451763.606777019
#Sta/Elev= 30
       0 1023.06    34.7 1011.02    48.3  998.18    64.7   989.1    91.1  982.31
   150.3   957.1   259.6  939.03   278.7  926.01   292.9  909.05   330.1  876.92
   379.2  850.18     407  838.37   459.3  830.86   576.1  829.57   595.2  823.45
   674.8  820.64   691.3  816.22   707.9  815.62   781.2   816.2   804.1  821.07
   819.7  835.83   829.9  838.89  1016.4  849.99  1048.4   856.6    1075  855.98
  1088.3  860.56  1138.2  865.81  1238.1  892.12  1331.3  909.83  1385.2  942.35
#Mann= 5 ,-1,0
       0      .1       0   691.3    .045       0   781.2      .1       0
  940.53     .05       0  990.53      .1       0
Bank Sta=691.3,781.2
XS Rating Curve= 0 ,0
Exp/Cntr(USF)=0,0
Exp/Cntr=0.3,0.1

Type RM Length L Ch R = 1 ,123372  ,523.5,500.4,468.7
XS GIS Cut Line= 6
1663714.80498414451820.2830089781664460.69850548451902.317293733
1664539.84237605451896.2188807281664746.76879947451893.975446895
1664972.61939764451897.619796559 1665200.9168413451911.595162317
#Sta/Elev= 30
       0 1149.02    44.4 1143.25   140.1 1120.31   225.9 1093.71   295.3 1063.73
   311.8 1052.27   338.2 1026.53   371.2 1009.98     391  992.05   414.1  980.37
   433.9  959.72   447.1   941.4   483.4  904.65   519.7  877.58     589     838
   635.3  826.91   656.2815.3433   730.7  814.22   748.4815.3447   786.9  820.86
   800.1  830.56   809.9  832.61   990.5  842.25  1108.6  858.25  1138.1  857.98
  1318.6  895.27  1344.9  895.47    1381  903.11  1423.8  920.48  1491.4  956.45
#Mann= 5 ,-1,0
       0      .1       0   656.2    .045       0   748.4      .1       0
  938.52     .05       0 1028.52      .1       0
Bank Sta=656.2,748.4
XS Rating Curve= 0 ,0
Exp/Cntr(USF)=0,0
Exp/Cntr=0.3,0.1

Type RM Length L Ch R = 1 ,122872  ,500.9,500,501.1
XS GIS Cut Line= 6
1663977.12827839452613.567183554 1664090.9367778452618.655099899
1664352.24957539452482.7718414811664579.59885822452364.550293148
1665156.98254597452064.3097518981665245.35769731452018.354791313
#Sta/Elev= 30
       0 1020.97    57.4 1011.56   113.9  992.34   172.3  997.29   225.1  991.64
   272.2  994.47   364.6  987.93   444.5  976.89   457.1  970.14   468.2  958.89
   475.6  947.98   509.7  918.41   532.7  901.75   553.2  883.03   571.7  861.89
   610.9  839.03     642  828.28   667.9  825.68  688.19814.8442   756.6  813.84
   797.4814.8058   823.5  828.38   857.6   835.5  1026.5  837.41  1165.6  848.36
  1207.9  846.52  1263.2  860.99  1314.9   888.4  1345.8  899.63  1415.1  915.85
#Mann= 4 ,-1,0
       0      .1       0  688.19    .045       0   797.4     .08       0
   804.7      .1       0
Bank Sta=688.19,797.4
XS Rating Curve= 0 ,0
Exp/Cntr(USF)=0,0
Exp/Cntr=0.3,0.1

Type RM Length L Ch R = 1 ,122372  ,456.7,500,561.1
XS GIS Cut Line= 6
 1664025.2459643452716.0899443921664187.17247772452823.700293481
1664334.31916505452910.4396213141664462.94193931452958.643593147
1664558.08709022452932.9139858041665459.19814889452484.219673231
#Sta/Elev= 30
       0 1008.04    73.9  986.11   137.8  953.43   230.5   918.4   288.8  909.67
   367.2  891.07   404.2  886.49   472.5  871.62   500.5  870.32   582.1     877
   682.1  873.34   760.4  852.42   808.1  828.01   848.3  824.94   859.4  815.26
   877.8  813.03   994.4815.3228  1006.1  820.16  1035.5     818  1064.8  820.16
  1108.8  844.83  1141.9  847.54  1163.7  853.02  1244.7  882.63  1325.3  895.64
  1427.8  942.86  1457.3  951.09  1512.2  978.53    1575  995.12  1607.8  995.14
#Mann= 3 ,-1,0
       0      .1       0   859.4    .045       0   994.4      .1       0
Bank Sta=859.4,994.4
XS Rating Curve= 0 ,0
Exp/Cntr(USF)=0,0
Exp/Cntr=0.3,0.1

Type RM Length L Ch R = 1 ,121872  ,431.8,471.8,511.1
XS GIS Cut Line= 6
1664029.27056256452727.4196461441664495.13905339453049.281535223
1664622.48131838 453114.189869971664715.80199789453143.687514395
1664792.53675255453186.4531769011665474.97042705453650.731119722
#Sta/Elev= 30
       0 1005.39    64.8  985.83   129.3  952.48   212.2  918.89   322.1   900.3
   392.9  881.95   498.4  862.92   620.1  862.51   715.4  837.25   965.2  823.34
   984.9 813.188   994.4   811.6 1068.68813.1281  1093.2  827.46  1132.9  829.65
  1163.6  840.07  1204.4  866.44  1220.2  886.37  1244.5  904.21  1303.5  971.29
  1327.1  983.53  1396.9  996.85  1414.6 1013.14  1442.9 1029.95  1474.1 1067.29
  1513.5 1090.18  1561.4 1103.27  1589.3 1118.41  1628.9 1124.73  1720.4 1167.27
#Mann= 3 ,-1,0
       0      .1       0   984.9    .045       0 1068.68      .1       0
Bank Sta=984.9,1068.68
XS Rating Curve= 0 ,0
Exp/Cntr(USF)=0,0
Exp/Cntr=0.3,0.1

Type RM Length L Ch R = 1 ,121400  ,526.3,535.1,542.8
XS GIS Cut Line= 3
1664015.37699297452751.8089992151664518.76348908453182.547448227
1664518.76348908454189.188151473
#Sta/Elev= 30
       0 1004.43      77  979.49   123.8  953.19   204.5  918.76   297.2  902.98
   433.6  869.14   673.1  838.49   873.3  830.84   892.9  819.53   932.1811.5977
   942.2  810.47  1011.5811.5788  1047.1  829.04  1125.9  843.39  1157.4  860.89
  1181.7  869.45  1309.6  976.22  1332.6  989.65  1371.9 1001.41  1385.1 1016.37
  1401.5 1026.53  1424.4 1064.88  1438.8 1075.22  1467.1 1086.39  1493.3 1086.78
  1526.1 1105.01  1552.4  1110.5  1581.9 1124.31  1631.1 1136.25  1669.2 1153.71
#Mann= 3 ,-1,0
       0      .1       0   932.1    .045       0  1011.5      .1       0
Bank Sta=932.1,1011.5
XS Rating Curve= 0 ,0
Exp/Cntr(USF)=0,0
Exp/Cntr=0.3,0.1

Type RM Length L Ch R = 1 ,120865  ,516.1,514.3,512
XS GIS Cut Line= 6
1663959.37437689452724.1076449011664055.42897481452839.736350641
 1664070.8324873452942.5114075541663947.51088355453740.854955226
1663902.54771888454031.9340974841663887.34105639454130.375829726
#Sta/Elev= 30
       0 1016.24    46.8 1009.65   127.8  985.12   199.2  950.68   232.7  941.87
   285.4  918.44   402.3   877.9   504.5  830.37   534.3  825.95   640.6  826.33
  665.14811.2813   703.7  811.27   819.9  809.79   832.7  810.41   846.5  817.22
     873   820.7   879.7  824.09   916.2  858.19   942.9  870.78   959.3  892.32
  1005.8  940.17  1025.7  953.11  1072.2  965.06  1118.7  983.69  1184.4  982.87
  1198.4  988.42  1317.9 1004.06  1367.7 1023.72  1417.5 1031.16  1456.2  1044.2
#Mann= 3 ,-1,0
       0      .1       0  665.14    .045       0   703.7      .1       0
Bank Sta=665.14,703.7
XS Rating Curve= 0 ,0
Exp/Cntr(USF)=0,0
Exp/Cntr=0.3,0.1

Type RM Length L Ch R = 1 ,120351  ,570.5,521.5,474.6
XS GIS Cut Line= 6
1663474.75994295453055.4448274211663507.59632709453256.045803289
1663487.53739405453483.2580294761663505.36905131453668.554574892
1663579.55853547453880.2263956371663765.59458072454111.214450732
#Sta/Elev= 30
       0  976.43    16.5  956.86    39.8  934.73    53.1  914.06    79.7  891.01
   116.3  853.65   149.5  830.66   189.4  818.66     206  817.04     218809.0143
   232.2  808.12  311.17809.0713   393.8  809.39   430.1  824.36   551.4  832.99
   742.6  866.16   762.2   871.7   787.7   883.6   812.6  890.51   826.8  891.34
     841  896.51   873.6  901.37   911.2  912.41     926  913.27   974.6   938.3
  1032.8  963.22  1052.7  975.58  1069.7  982.53  1097.9  991.12  1139.4  995.79
#Mann= 5 ,-1,0
       0      .1       0     218    .045       0  311.17      .1       0
  316.51     .08       0  406.51      .1       0
Bank Sta=218,311.17
XS Rating Curve= 0 ,0
Exp/Cntr(USF)=0,0
Exp/Cntr=0.3,0.1

Type RM Length L Ch R = 1 ,119829  ,522.3,500,490.2
XS GIS Cut Line= 6
1662844.74963763453511.5663718131663402.80331156453764.018950894
1663483.77755906 453820.060505481663553.91718255453904.092489645
1663649.59940588454006.0643985571663759.18416047 454117.18097423
#Sta/Elev= 30
       0    1028    13.1 1019.36    27.5 1002.48    41.9   995.4    56.3  991.75
    79.2  976.24    99.5  948.82   142.8  912.03   153.5  898.44     180  878.33
   190.6  866.09     222  846.96   234.5  829.93   254.4  810.59   276.2806.4384
   322.8  806.05   329.8806.4346   369.6  810.04   391.2  818.25     420  823.28
   470.4  824.51   625.6  839.95   694.5  861.71   735.9  868.35   810.6  890.19
   875.8  902.36   973.1   945.1  1033.4  977.93  1071.9  989.15  1116.3  996.81
#Mann= 4 ,-1,0
       0      .1       0   276.2    .045       0   329.8     .08       0
  336.25      .1       0
Bank Sta=276.2,329.8
XS Rating Curve= 0 ,0
Exp/Cntr(USF)=0,0
Exp/Cntr=0.3,0.1

Type RM Length L Ch R = 1 ,119329  ,483.6,498.4,504.7
XS GIS Cut Line= 6
1662826.16535722454149.7665389781662912.43027656454135.116961971
1663084.95978713454105.8171518151663530.14852931454030.213956565
1663637.71524331454069.1249679771663753.24191514 454148.71142298
#Sta/Elev= 30
       0  938.68      21  937.41    37.6  931.54    70.9  899.54    87.5  876.34
   102.1  861.82   110.8  844.62   114.2  840.21   127.5  832.54   147.6  817.41
   157.4  808.16   168.1804.6464   190.7  803.53   223.9804.6511   250.6   806.8
   277.2  814.38   290.5  814.87   303.8  820.83   363.8  823.79   446.9  834.49
   463.6  838.93   523.5  846.01   666.6  878.81   720.1  897.85     762  916.37
   800.3  940.89   840.2  959.62     872  981.61   911.9  989.11   968.7 1005.26
#Mann= 3 ,-1,0
       0      .1       0   168.1    .045       0   223.9      .1       0
Bank Sta=168.1,223.9
XS Rating Curve= 0 ,0
Exp/Cntr(USF)=0,0
Exp/Cntr=0.3,0.1

Type RM Length L Ch R = 1 ,118831  ,436.2,501.6,538
XS GIS Cut Line= 6
1662778.37673889454440.9916783121662892.38372873454569.768323645
1662980.11878946454591.3250390591663054.65702622454602.616355062
 1663154.3815643454610.7065619831663410.32724664454623.190788984
#Sta/Elev= 30
       0  877.46    55.4   866.7   103.3  855.59   160.6  843.72   209.6  835.62
   271.6  821.07     286  816.78   300.1   811.4     310  809.44     320  805.82
   329.8  803.54   362.9  802.94   413.2803.5509   418.9  805.24   429.2   811.2
   441.9  816.79   451.8  818.96   464.9  818.87   468.2  819.64   478.1  824.34
   484.6  826.05     524   831.6   537.2  835.53   563.5  851.77   580.5  865.28
   609.4  881.88   635.7  899.39   642.3  903.03   675.1  917.44     694  929.27
#Mann= 3 ,-1,0
       0      .1       0   329.8    .045       0   413.2      .1       0
Bank Sta=329.8,413.2
XS Rating Curve= 0 ,0
Exp/Cntr(USF)=0,0
Exp/Cntr=0.3,0.1

Type RM Length L Ch R = 1 ,118329  ,478.5,499.1,511.6
XS GIS Cut Line= 6
1662715.77417381454503.4541518091662767.17859855454694.693598732
1662763.71666323454800.274752393 1662762.1756558454875.459641397
 1662767.4315508454975.3213183131662780.90035589455231.217131972
#Sta/Elev= 30
       0  865.99    39.5   858.9    59.8  851.23    80.2  845.53   161.8  832.18
   225.4   828.3   281.2  829.08   310.7  826.98   323.8  824.36   327.1  822.35
     337  812.47   346.8  807.57   353.4   806.3   379.6  805.46   398.4802.2382
   412.5  801.16   456.8802.2511   474.9   812.4   484.7  814.48     511  823.85
   524.2  825.67   550.4  832.87   560.3   838.2   593.2  859.87     626  888.03
   635.9  898.57     649  915.93   681.9  946.27   697.3  962.72   735.1  994.39
#Mann= 3 ,-1,0
       0      .1       0   398.4    .045       0   456.8      .1       0
Bank Sta=398.4,456.8
XS Rating Curve= 0 ,0
Exp/Cntr(USF)=0,0
Exp/Cntr=0.3,0.1

Type RM Length L Ch R = 1 ,117830  ,508.8,500.8,491.2
XS GIS Cut Line= 6
1662469.24550925454252.9412022711662449.23718214454554.566336502
1662373.77649823454657.5480037331662327.79233822454716.889748558
1662269.69698197454782.9798394741662138.85013081454923.936250478
#Sta/Elev= 30
       0  929.66    29.5  925.51    42.7  922.52    88.3  916.71   108.4  910.97
     163  885.88   210.3  871.04   226.8  864.33   237.1  859.61   249.8  851.24
   276.1  841.18   304.3  822.03   314.6  808.27     333801.8214     370  800.93
   447.2801.7995   465.8  808.84   512.8  813.58   542.4  821.48   564.3  823.68
   603.8     832   635.1  840.24   697.6  860.03   715.6  869.37   738.1  886.83
   745.1  893.47   760.5   911.9   763.7  914.75   775.3  919.61   785.4  926.29
#Mann= 3 ,-1,0
       0      .1       0     333    .045       0   447.2      .1       0
Bank Sta=333,447.2
XS Rating Curve= 0 ,0
Exp/Cntr(USF)=0,0
Exp/Cntr=0.3,0.1

Type RM Length L Ch R = 1 ,117329  ,475.9,500.1,509
XS GIS Cut Line= 6
1662154.71722506454005.0355292261662067.95689988454174.818982303
 1662028.2775173454252.8230913881661994.52003889454319.806225151
 1661950.7953888454409.7404284781661796.73598564454727.487168312
#Sta/Elev= 30
       0  979.38    16.7  968.92    30.7  964.36    90.4  930.52   113.5  920.06
     155  906.42   200.9  894.63     223  884.51     277  853.33     337  808.37
   342.9  802.58   354.2800.6467   406.4  800.29   438.3800.6439   472.1  807.93
     545  810.71     607  829.28   636.2  847.14   647.3  855.94     667  866.19
   679.9  880.17   705.4  897.96   716.1  910.52     731  920.44   738.2  930.04
   753.1  938.11   768.1  956.58   774.7  962.28   785.6  969.89   806.3  977.68
#Mann= 3 ,-1,0
       0      .1       0   354.2    .045       0   438.3      .1       0
Bank Sta=354.2,438.3
XS Rating Curve= 0 ,0
Exp/Cntr(USF)=0,0
Exp/Cntr=0.3,0.1

Type RM Length L Ch R = 1 ,116829  ,498.6,500,502.1
XS GIS Cut Line= 6
1661950.23206972453791.1888440551661882.04716672453865.559430227
1661810.07651013453931.7472899711661455.99257264454177.920354053
1661384.14921239454227.8684168911661197.07679376454352.414919218
#Sta/Elev= 30
       0  973.46    83.3  949.01   180.8  911.59   226.6  885.94   255.4  872.29
   301.4  845.65   335.9  828.94   363.3  810.79     394  808.36   410.4  803.14
   429.3  800.79   461.2799.1569   470.3  798.09   521.4799.1536   530.7  802.42
   540.1  808.31   582.6  818.66   626.2  838.06     658  849.93     698  878.44
   714.1  887.11   733.8  903.58   762.5  918.61     795  946.58   844.2   970.7
   863.1  991.72   879.7 1005.68   903.8 1014.96   924.4  1017.9   942.2 1025.32
#Mann= 3 ,-1,0
       0      .1       0   461.2    .045       0   521.4      .1       0
Bank Sta=461.2,521.4
XS Rating Curve= 0 ,0
Exp/Cntr(USF)=0,0
Exp/Cntr=0.3,0.1
